HEC-RAS study E100-00-00.prj: E100-00-00

--- E100-00-00.g02 (geometry) --- (continued)

Type RM Length L Ch R = 3 ,99176.0 ,,,
BEGIN DESCRIPTION:
LAKEVIEW
Structure ID: E100-00-00-50
END DESCRIPTION:
Bridge Culvert--1,0,-1,-1, 0
Deck Dist Width WeirC Skew NumUp NumDn MinLoCord MaxHiCord MaxSubmerge Is_Ogee
10,32,2.6,0, 60, 60, , , 0.95, 0, ,,,
  1702.5  1782.6  1832.6  2262.6  2342.6  2392.6  2622.6  2752.6  2812.6  2832.6
  2932.6  3302.6  3342.6  3832.6  3902.6  3972.6  4142.6  4462.6  4702.6  4722.6
  4809.4  4901.2 4952.69  4952.8  4954.2  4957.7 5079.69  5079.8  5086.7 5086.81
  5116.4    5182  5348.5  5368.5  5388.5  5408.5    5960    6170    6350    6390
    6440    7010    7340    7450    7490    7530    7570    7610    7750    7820
    8440    8490    8870    9620    9640    9680    9690    9710    9720  9758.5
   109.8   108.8   106.5   104.1   103.1   104.9   105.2   103.8   101.4   101.4
   103.9   103.4   102.5   102.7   101.8   102.9   100.7  100.51   99.71   99.11
   99.15   99.46  100.42  102.86  102.86  102.85  102.64  102.64  102.63   99.73
   99.21   99.56   98.81   98.73   98.71   99.81   102.7   102.1   103.2   102.1
   104.3   104.2   105.8   105.6     105   105.3   104.6   106.4   106.1   104.4
     106   104.7   105.9   105.5   105.1     106   107.2   115.2   116.7   118.4
   109.8   108.8   106.5   104.1   103.1   104.9   105.2   103.8   101.4   101.4
   103.9   103.4   102.5   102.7   101.8   102.9   100.7   100.5    99.7    99.1
   99.04   99.28  100.41  100.41  100.39   98.45   98.24   97.89    98.9   98.91
    99.2   99.55    98.8    98.2    98.7    99.8   102.7   102.1   103.2   102.1
   104.3   104.2   105.8   105.6     105   105.3   104.6   106.4   106.1   104.4
     106   104.7   105.9   105.5   105.1     106   107.2   115.2   116.7   118.4
  1702.5  1782.6  1832.6  2262.6  2342.6  2392.6  2622.6  2752.6  2812.6  2832.6
  2932.6  3302.6  3342.6  3832.6  3902.6  3972.6  4142.6  4462.6  4702.6  4722.6
  4809.4  4901.2 4952.69  4952.8 4952.91  4954.2 5079.69  5079.8  5086.7 5086.81
  5116.4    5182  5348.5  5368.5  5388.5  5408.5    5960    6170    6350    6390
    6440    7010    7340    7450    7490    7530    7570    7610    7750    7820
    8440    8490    8870    9620    9640    9680    9690    9710    9720  9758.5
   109.8   108.8   106.5   104.1   103.1   104.9   105.2   103.8   101.4   101.4
   103.9   103.4   102.5   102.7   101.8   102.9   100.7  100.51   99.71   99.11
   99.15   99.46  100.42  102.86  102.86  102.86  102.64  102.64  102.63   99.73
   99.21   99.56   98.81   98.73   98.71   99.81   102.7   102.1   103.2   102.1
   104.3   104.2   105.8   105.6     105   105.3   104.6   106.4   106.1   104.4
     106   104.7   105.9   105.5   105.1     106   107.2   115.2   116.7   118.4
   109.8   108.8   106.5   104.1   103.1   104.9   105.2   103.8   101.4   101.4
   103.9   103.4   102.5   102.7   101.8   102.9   100.7   100.5    99.7    99.1
   99.04   99.28  100.41  100.41   98.45   98.45   98.24   97.89    98.9   98.91
    99.2   99.55    98.8    98.2    98.7    99.8   102.7   102.1   103.2   102.1
   104.3   104.2   105.8   105.6     105   105.3   104.6   106.4   106.1   104.4
     106   104.7   105.9   105.5   105.1     106   107.2   115.2   116.7   118.4
Pier Skew, UpSta & Num, DnSta & Num=  ,4989.8, 2 ,4989.8, 2 , 0 , 0 , 0 ,,
       2       2
   82.53    99.4
       2       2
   81.44    99.4
Pier Skew, UpSta & Num, DnSta & Num=  ,5019.9, 2 ,5019.9, 2 , 0 , 0 , 0 ,,
       2       2
   84.34   99.35
       2       2
   83.25   99.35
Pier Skew, UpSta & Num, DnSta & Num=  ,5050, 2 ,5050, 2 , 0 , 0 , 0 ,,
       2       2
   86.98   99.29
       2       2
   85.89   99.29
BR Coef= 1 , 1 , 0 ,1.25, 0 ,,,0.8,-1,2,0,
WSPro=,,,, 1 ,,,, 0 ,,,, 0 ,,,,-1 ,-1 ,-1 , 0 , 0 , 0 , 0 , 0
BR U #Sta/Elev= 99
  1702.5   109.8  1702.6   109.8  1782.6   108.8  1832.6   106.5  2262.6   104.1
  2342.6   103.1  2392.6   104.9  2622.6   105.2  2752.6   103.8  2812.6   101.4
  2832.6   101.4  2932.6   103.9  3302.6   103.4  3342.6   102.5  3832.6   102.7
  3902.6   101.8  3972.6   102.9  4142.6   100.7  4267.1  100.62  4462.6   100.5
  4567.6  100.15  4702.6    99.7  4722.6    99.1  4809.4   99.04  4861.4   99.38
  4884.3   99.53  4901.2   99.28  4913.7   99.54  4915.1   99.57  4942.8  100.52
  4943.8  100.51 4952.69  100.41  4952.8  100.41 4952.91   100.4  4954.2  100.39
 4957.61   98.47  4957.7   98.42  4958.9   97.75    4961   96.23  4989.8   86.47
  4990.2    86.1  4990.4    84.4  4990.6   83.53  5001.2    83.4  5007.7   83.56
  5009.5    84.4  5013.5   85.38  5018.1   87.03  5019.9   85.19  5032.6   87.09
  5047.3   87.53    5050   88.25  5078.6   97.71 5079.69   97.87  5079.8   97.89
 5086.59   98.88  5086.7    98.9 5086.81   98.91  5089.3   99.28  5116.4    99.2
    5131   99.28    5182   99.55    5185   99.53  5216.8   99.32  5234.4   99.21
  5279.1   99.05  5348.5    98.8  5368.5    98.2  5388.5    98.7  5399.1   99.28
  5408.5    99.8  5628.1  100.94    5660   101.1  5955.3  102.67    5960   102.7
    6170   102.1    6350   103.2    6390   102.1    6440   104.3    7010   104.2
    7340   105.8    7450   105.6    7490     105    7530   105.3    7570   104.6
    7610   106.4    7750   106.1    7820   104.4    8440     106    8490   104.7
  8797.2  105.67    8870   105.9    9620   105.5    9640   105.1    9680     106
    9690   107.2    9710   115.2    9720   116.7  9758.5   118.4
BR U #Mann= 7
  1702.5     .99  1702.6     .08  4943.8     .04  4954.2     .04  5089.3     .08
  8797.2      .1  9758.5     .99
BR U Banks=4954.2,5089.3
BR D #Sta/Elev= 99
  1702.5   109.8  1702.6   109.8  1782.6   108.8  1832.6   106.5  2262.6   104.1
  2342.6   103.1  2392.6   104.9  2622.6   105.2  2752.6   103.8  2812.6   101.4
  2832.6   101.4  2932.6   103.9  3302.6   103.4  3342.6   102.5  3832.6   102.7
  3902.6   101.8  3972.6   102.9  4142.6   100.7  4267.1  100.62  4462.6   100.5
  4567.6  100.15  4702.6    99.7  4722.6    99.1  4809.4   99.04  4861.4   99.38
  4884.3   99.53  4901.2   99.28  4913.7   99.54  4915.1   99.57  4942.8  100.52
  4943.8  100.51 4952.69  100.41  4952.8  100.41 4952.91   100.4  4954.2    99.3
 4957.61   97.38  4957.7   97.33  4958.9   96.66    4961   95.14  4989.8   85.38
  4990.2   85.01  4990.4   83.31  4990.6   82.44  5001.2   82.31  5007.7   82.47
  5009.5   83.31  5013.5   84.29  5018.1   85.94  5019.9    84.1  5032.6      86
  5047.3   86.44    5050   87.16  5078.6   96.62 5079.69   97.87  5079.8   97.89
 5086.59   98.88  5086.7    98.9 5086.81   98.91  5089.3   99.28  5116.4    99.2
    5131   99.28    5182   99.55    5185   99.53  5216.8   99.32  5234.4   99.21
  5279.1   99.05  5348.5    98.8  5368.5    98.2  5388.5    98.7  5399.1   99.28
  5408.5    99.8  5628.1  100.94    5660   101.1  5955.3  102.67    5960   102.7
    6170   102.1    6350   103.2    6390   102.1    6440   104.3    7010   104.2
    7340   105.8    7450   105.6    7490     105    7530   105.3    7570   104.6
    7610   106.4    7750   106.1    7820   104.4    8440     106    8490   104.7
  8797.2  105.67    8870   105.9    9620   105.5    9640   105.1    9680     106
    9690   107.2    9710   115.2    9720   116.7  9758.5   118.4
BR D #Mann= 6
  1702.5     .99  1702.6     .08  4943.8     .04  4954.2     .04  5089.3     .08
  8797.2      .1
BR D Banks=4954.2,5089.3
BC Design=,, 0 ,, 0 ,,,,,,
BC HTab HWMax=118.4
BC Use User HTab Curves=0
BC User HTab FreeFlow(D)= 0

Type RM Length L Ch R = 1 ,99154.0 ,118.6,110,108.3
BEGIN DESCRIPTION:
Downstream Section of Bridge/Culvert/Weir
END DESCRIPTION:
XS GIS Cut Line= 5
      3061706.03     13888918.71       3059730.7     13886350.84
      3059634.79     13886253.06       3059311.5     13885769.06
      3056330.78     13882951.05
#Sta/Elev= 30
  1702.5   109.8  1702.6   109.8  1832.6   106.5  2342.6   103.1  2622.6   105.2
  2812.6   101.4  2932.6   103.9  3972.6   102.9  4722.6    99.1  4943.8  100.51
  4954.2   99.28  4989.8   85.36  4990.6   82.42  5001.2   82.29  5018.1   85.92
  5019.9   84.08  5047.3   86.42 5079.69   97.87  5089.3   99.28  5368.5    98.2
    5960   102.7    7570   104.6    7610   106.4    7820   104.4  8797.2  105.67
    9640   105.1    9680     106    9690   107.2    9710   115.2  9758.5   118.4
#Mann= 7 ,-1 , 0
  1702.5     .99       0  1702.6     .08       0  4943.8     .04       0
  4954.2     .04       0  5089.3     .08       0  8797.2      .1       0
  9758.5     .99       0
#XS Ineff= 3 ,-1
    2000    2940   104.1  5089.7    8000    98.8    4000  4949.8    98.8
Permanent Ineff=
       F       F       F
Bank Sta=4954.2,5089.3
XS Rating Curve= 0 ,0
Exp/Cntr=0.5,0.3

Type RM Length L Ch R = 1 ,99044.  ,414.1,480,473.1
BEGIN DESCRIPTION:
Lakeview - D\S - XS 1
END DESCRIPTION:
XS GIS Cut Line= 5
      3061480.08     13888445.56      3059809.94     13886274.44
      3059714.03     13886176.65      3059390.74     13885692.65
      3056410.02     13882874.65
#Sta/Elev= 30
  2197.4  105.15  2367.4  105.32  2497.4  102.11  2587.4  103.89  2657.4  101.51
  2727.4  103.82  2997.4  104.38  3747.4   99.86  3947.4  102.53  4537.4   98.56
  4917.4  100.77  4946.6   97.34  4986.6   86.85 4988.71   83.27 4999.69   82.07
 5011.08   83.72  5046.6   95.81  5073.6   99.55  5303.6   98.31  5985.6  103.48
  6585.6  104.42  6715.6  102.63  7525.6  106.18  7695.6  103.97  7735.6   106.6
  9225.6  105.56  9575.6  105.35  9615.6  108.11  9635.6  114.28  9757.5     117
#Mann= 4 ,-1 , 0
  2197.4     .08       0  4917.4     .04       0  5073.6     .08       0
  9225.6      .1       0
#XS Ineff= 2 , 0
       0    3000  104.38               0
Permanent Ineff=
       F       F
Bank Sta=4917.4,5073.6
XS Rating Curve= 0 ,0
Exp/Cntr=0.3,0.1

Type RM Length L Ch R = 1 ,98564.0 ,720.8,891,906.7
BEGIN DESCRIPTION:
Cross Section E100-00-00-X71
END DESCRIPTION:
XS GIS Cut Line= 4
      3061644.17     13888662.78      3060224.07     13886094.76
      3060093.81     13885814.94      3056968.62     13882679.06
#Sta/Elev= 30
  1923.5   108.6  2123.5   103.8  2433.5   104.5  2613.5   101.8  2973.5   103.8
  3063.5   101.4  3233.5   103.9  3513.5    99.9  4163.5      98  4935.9   99.65
    4937   99.64  4960.3   89.89    4983   86.99  4993.1   81.12  5007.3   81.51
  5046.2   97.21  5049.4   97.18    5078    99.2  5596.7   101.2  5736.7    99.7
  6096.7   102.6  6176.7   100.4  6366.7   103.4  6666.7   101.6  6846.7   103.8
  8160.1  104.79  9476.7   104.9  9506.7   105.8  9546.7   114.2  9593.9   112.7
#Mann= 7 ,-1 , 0
  1923.5     .08       0  4935.9     .04       0    4937     .04       0
  5046.2     .04       0  5049.4     .08       0  8160.1      .1       0
  9593.9     .99       0
#XS Ineff= 2 , 0
       0  3233.5   103.9  6096.7       0   102.6
Permanent Ineff=
       F       F
Bank Sta=4937,5046.2
XS Rating Curve= 0 ,0
Exp/Cntr=0.3,0.1

Type RM Length L Ch R = 1 ,97673.  ,111.7,102,101
BEGIN DESCRIPTION:
Equador Drive - U\S - XS 4
END DESCRIPTION:
XS GIS Cut Line= 4
      3061485.71     13888292.58      3060956.39     13885735.09
      3060928.93     13885662.02      3059010.23     13881603.98
#Sta/Elev= 30
  2345.9  104.88  2805.9  103.88  2955.9   100.6  3315.9  102.68  3365.9  100.45
  3445.9  102.82  3785.9   99.55  3885.9  100.94  4925.9   98.66  4945.9   96.78
 4998.21   80.03 5009.01    81.2  5045.6   95.25  5075.6   98.69  5625.6   99.18
  5685.6   97.18  5995.6  100.68  6125.6   98.47  6855.6     102  7055.6   100.5
  7135.6  100.76  7205.6   90.33  7315.6   89.89  7335.6   92.04  7365.6   99.13
  7395.6  101.23  8285.6  100.95  8615.6  104.24  9275.6  101.08  9528.3  104.51
#Mann= 5 ,-1 , 0
  2345.9     .08       0  4925.9     .04       0  5075.6     .08       0
  7055.6     .05       0  8285.6     .08       0
#XS Ineff= 2 , 0
       0                    6240       0     104
Permanent Ineff=
       F       F
#Block Obstruct= 1 ,-1
 7131.28 7434.36  100.91
Bank Sta=4925.9,5075.6
XS Rating Curve= 0 ,0
Exp/Cntr=0.5,0.3

Type RM Length L Ch R = 1 ,97571.0 ,27,25,24.2
BEGIN DESCRIPTION:
Upstream Section of Bridge/Culvert/Weir
END DESCRIPTION:
XS GIS Cut Line= 4
      3061663.13     13888656.16      3061049.78     13885692.64
      3061022.32     13885619.57      3059103.61     13881561.53
#Sta/Elev= 30
  1935.1  108.71  2875.1  103.41  2905.1  101.21  3005.1  104.21  3265.1  104.01
  3485.1   99.91  3695.1  101.31  3735.1   99.71  4155.1   98.61  4936.5   98.21
    4942   98.42  4974.2   85.78  4998.8   79.91  5009.8   81.18  5029.2   91.47
  5048.2    98.6  5063.4  100.22  5068.9   99.97  5155.9   97.88  5569.5   99.31
  5669.5   96.91  5959.5  100.51  6099.5   98.41  6489.5  100.91  7071.1  100.91
  8251.3  100.95  8659.5  103.01  9189.5  102.71  9269.5  100.91  9528.3  104.51
#Mann= 7 ,-1 , 0
  1935.1     .08       0  4936.5     .04       0    4942     .04       0
  5063.4     .04       0  5068.9     .08       0  7071.1     .05       0
  8251.3     .08       0
#XS Ineff= 3 ,-1
    6250    9515     104  5057.9    6250    99.9    2500  4936.2    97.8
Permanent Ineff=
       F       F       F
Bank Sta=4942,5063.4
XS Rating Curve= 0 ,0
Exp/Cntr=0.5,0.3

Type RM Length L Ch R = 3 ,97558.0 ,,,
BEGIN DESCRIPTION:
EQUADOR DRIVE
Structure ID: E100-00-00-49
END DESCRIPTION:
Bridge Culvert--1,0,-1,-1, 0
Deck Dist Width WeirC Skew NumUp NumDn MinLoCord MaxHiCord MaxSubmerge Is_Ogee
10,6,2.6,0, 60, 60, , , 0.95, 0, ,,,
  1935.1  2875.1  2905.1  2935.1  2965.1  3005.1  3025.1  3265.1  3485.1  3695.1
  3715.1  3735.1  3915.1  4115.1  4155.1  4265.1  4515.1  4846.5    4890  4928.8
    4942 4946.19  4946.3  4998.8 5048.96 5049.07  5063.4  5065.8    5066 5066.11
  5101.5  5155.9  5214.5  5319.5  5559.5  5569.5  5669.5  5686.9  5749.5  5959.5
  6029.5  6069.5  6099.5  6131.2  6489.5  6529.5  6869.5  6999.5  7089.5  7099.5
  7429.5  7509.5  8129.5  8329.5  8379.5  8659.5  8739.5  9189.5  9269.5  9528.3
  108.71  103.41  101.21  101.41  103.41  104.21  104.01  104.01   99.91  101.31
  100.71   99.71  101.01   99.71   98.61   99.81   98.31   97.58   97.55   98.68
   98.96   99.04  102.54  103.63  104.45  104.45  104.69  104.73   104.7   101.2
   98.69   98.59    98.2   97.81   98.91   99.31   97.02   97.37   99.01  100.51
  100.41   98.55   98.67    98.8  100.91  100.21  101.81  100.91  100.91  100.11
  101.31  100.81  102.11  100.21  101.81  103.01  102.41  102.71  100.91  104.51
  108.71  103.41  101.21  101.41  103.41  104.21  104.01  104.01   99.91  101.31
  100.71   99.71  101.01   99.71   98.61   99.81   98.31   97.49   97.29   97.92
   98.42   96.95   96.95   98.04   98.86   98.69  100.22  100.11   100.1   100.1
   98.56   97.88    98.2   97.81   98.91   99.31   96.91   97.37   99.01  100.51
  100.41   98.51   98.41   98.61  100.91  100.21  101.81  100.91  100.91  100.11
  101.31  100.81  102.11  100.21  101.81  103.01  102.41  102.71  100.91  104.51
  1935.1  2875.1  2905.1  2935.1  2965.1  3005.1  3025.1  3265.1  3485.1  3695.1
  3715.1  3735.1  3915.1  4115.1  4155.1  4265.1  4515.1  4846.5    4890  4928.8
    4942 4946.19  4946.3  4998.8 5048.96 5049.07  5063.4  5065.8    5066 5066.11
  5101.5  5155.9  5214.5  5319.5  5559.5  5569.5  5669.5  5686.9  5749.5  5959.5
  6029.5  6069.5  6099.5  6131.2  6489.5  6529.5  6869.5  6999.5  7089.5  7099.5
  7429.5  7509.5  8129.5  8329.5  8379.5  8659.5  8739.5  9189.5  9269.5  9528.3
  108.71  103.41  101.21  101.41  103.41  104.21  104.01  104.01   99.91  101.31
  100.71   99.71  101.01   99.71   98.61   99.81   98.31   97.58   97.55   98.68
   98.96   99.04  102.54  103.63  104.45  104.45  104.69  104.73   104.7   101.2
   98.69   98.59    98.2   97.81   98.91   99.31   97.02   97.37   99.01  100.51
  100.41   98.55   98.67    98.8  100.91  100.21  101.81  100.91  100.91  100.11
  101.31  100.81  102.11  100.21  101.81  103.01  102.41  102.71  100.91  104.51
  108.71  103.41  101.21  101.41  103.41  104.21  104.01  104.01   99.91  101.31
  100.71   99.71  101.01   99.71   98.61   99.81   98.31   97.49   97.29   97.92
   98.42   96.95   96.95   98.04   98.86   98.69  100.22  100.11   100.1   100.1
   98.56   97.88    98.2   97.81   98.91   99.31   96.91   97.37   99.01  100.51
  100.41   98.51   98.41   98.61  100.91  100.21  101.81  100.91  100.91  100.11
  101.31  100.81  102.11  100.21  101.81  103.01  102.41  102.71  100.91  104.51
Pier Skew, UpSta & Num, DnSta & Num=  ,4961.4, 2 ,4961.4, 2 , 0 , 0 , 0 ,,
       1       1
    90.6   98.27
       1       1
    90.9   98.57
Pier Skew, UpSta & Num, DnSta & Num=  ,4981.3, 2 ,4981.3, 2 , 0 , 0 , 0 ,,
       1       1
   83.68   98.69
       1       1
   83.98   98.99
Pier Skew, UpSta & Num, DnSta & Num=  ,5001.6, 2 ,5001.6, 2 , 0 , 0 , 0 ,,
       1       1
   79.18   99.09
       1       1
   79.48   99.39
Pier Skew, UpSta & Num, DnSta & Num=  ,5020.6, 2 ,5020.6, 2 , 0 , 0 , 0 ,,
       1       1
    85.6    99.4
       1       1
    85.9    99.7
Abutment Skew #Up #Dn= , 2 , 2
 4940.37 4984.77
   98.37   83.95
 4940.37 4984.77
   98.67   84.25
Abutment Skew #Up #Dn= , 2 , 2
 5004.27 5049.16
   80.56   98.86
 5004.27 5049.16
   80.86   99.16
BR Coef= 1 , 1 , 0 ,1.25, 0 ,,,0.8,0,2,0,
WSPro=,,,, 1 ,,,, 0 ,,,, 0 ,,,,-1 ,-1 ,-1 , 0 , 0 , 0 , 0 , 0
BR U #Sta/Elev= 99
  1935.1  108.71  2875.1  103.41  2905.1  101.21  2935.1  101.41  2965.1  103.41
  3005.1  104.21  3025.1  104.01  3265.1  104.01  3485.1   99.91  3695.1  101.31
  3715.1  100.71  3735.1   99.71  3915.1  101.01  4115.1   99.71  4155.1   98.61
  4265.1   99.81  4515.1   98.31  4527.5   98.28  4846.5   97.49    4848   97.48
  4888.9   97.27    4890   97.29  4928.8   97.92  4931.4   98.02  4936.5   98.21
 4940.48   98.36 4940.57   98.37    4942   98.42  4946.1   96.45 4946.19   96.41
  4946.3   96.36 4946.41   96.31  4948.3    95.4  4959.9   92.65  4966.9   88.91
  4974.2   85.78  4980.2   84.66  4983.3   84.79 4984.77   83.95  4986.8   82.79
  4988.8   82.56  4990.3   81.07  4991.1   80.59  4997.1   80.06  4998.8   79.91
 5004.27   80.56  5007.1    80.9  5007.2   80.21  5009.8   81.18  5012.5   83.24
  5022.2   87.55  5026.1   89.14  5029.2   91.47  5048.2    98.6 5048.96   98.68
 5049.07   98.69  5063.4  100.22  5065.8  100.11 5065.89  100.11    5066   100.1
 5066.11   100.1  5068.9   99.97  5081.9   99.37  5101.5   98.56  5102.8   98.51
  5155.9   97.88  5164.1   97.92  5214.5    98.2  5286.9   97.93  5319.5   97.81
  5559.5   98.91  5569.5   99.31  5669.5   96.91  5686.9   97.37  5749.5   99.01
  5959.5  100.51  6029.5  100.41  6069.5   98.51  6099.5   98.41  6131.2   98.61
  6489.5  100.91  6529.5  100.21  6869.5  101.81  6999.5  100.91  7071.1  100.91
  7089.5  100.91  7099.5  100.11  7429.5  101.31  7509.5  100.81  8129.5  102.11
  8251.3  100.95  8329.5  100.21  8379.5  101.81  8659.5  103.01  8739.5  102.41
  9189.5  102.71  9269.5  100.91  9299.5  101.31  9528.3  104.51
BR U #Mann= 8
  1935.1     .99  1935.1     .08  4936.5     .04    4942     .04  5063.4     .04
  5068.9     .08  7071.1     .05  8251.3     .08
BR U Banks=4942,5063.4
BR D #Sta/Elev= 99
  1935.1  108.71  2875.1  103.41  2905.1  101.21  2935.1  101.41  2965.1  103.41
  3005.1  104.21  3025.1  104.01  3265.1  104.01  3485.1   99.91  3695.1  101.31
  3715.1  100.71  3735.1   99.71  3915.1  101.01  4115.1   99.71  4155.1   98.61
  4265.1   99.81  4515.1   98.31  4527.5   98.28  4846.5   97.49    4848   97.48
  4888.9   97.27    4890   97.29  4928.8   97.92  4931.4   98.02  4936.5   98.21
 4940.48   98.36 4940.57   98.37    4942   98.72  4946.1   96.75 4946.19   96.71
  4946.3   96.66 4946.41   96.61  4948.3    95.7  4959.9   92.95  4966.9   89.21
  4974.2   86.08  4980.2   84.96  4983.3   85.09 4984.77   84.25  4986.8   83.09
  4988.8   82.86  4990.3   81.37  4991.1   80.89  4997.1   80.36  4998.8   80.21
 5004.27   80.86  5007.1    81.2  5007.2   80.51  5009.8   81.48  5012.5   83.54
  5022.2   87.85  5026.1   89.44  5029.2   91.77  5048.2    98.9 5048.96   98.98
 5049.07   98.99  5063.4  100.52  5065.8  100.11 5065.89  100.11    5066   100.1
 5066.11   100.1  5068.9   99.97  5081.9   99.37  5101.5   98.56  5102.8   98.51
  5155.9   97.88  5164.1   97.92  5214.5    98.2  5286.9   97.93  5319.5   97.81
  5559.5   98.91  5569.5   99.31  5669.5   96.91  5686.9   97.37  5749.5   99.01
  5959.5  100.51  6029.5  100.41  6069.5   98.51  6099.5   98.41  6131.2   98.61
  6489.5  100.91  6529.5  100.21  6869.5  101.81  6999.5  100.91  7071.1  100.91
  7089.5  100.91  7099.5  100.11  7429.5  101.31  7509.5  100.81  8129.5  102.11
  8251.3  100.95  8329.5  100.21  8379.5  101.81  8659.5  103.01  8739.5  102.41
  9189.5  102.71  9269.5  100.91  9299.5  101.31  9528.3  104.51
BR D #Mann= 7
  1935.1     .08  4936.5     .04    4942     .04  5063.4     .04  5068.9     .08
  7071.1     .05  8251.3     .08
BR D Banks=4942,5063.4
BC Design=,, 0 ,, 0 ,,,,,,
BC HTab HWMax=108.71
BC Use User HTab Curves=0
BC User HTab FreeFlow(D)= 0

Type RM Length L Ch R = 1 ,97546.0 ,91.5,101,102
BEGIN DESCRIPTION:
Downstream Section of Bridge/Culvert/Weir
END DESCRIPTION:
XS GIS Cut Line= 4
      3061687.23     13888653.17       3061073.4     13885687.36
      3061044.68     13885610.95      3059125.45     13881551.79
#Sta/Elev= 30
  1935.1  108.71  2875.1  103.41  2905.1  101.21  3005.1  104.21  3265.1  104.01
  3485.1   99.91  3695.1  101.31  3735.1   99.71  4155.1   98.61  4936.5   98.21
    4942   98.64  4974.2      86  4998.8   80.13  5009.8    81.4  5029.2   91.69
  5048.2   98.82  5063.4  100.44  5068.9   99.97  5155.9   97.88  5569.5   99.31
  5669.5   96.91  5959.5  100.51  6099.5   98.41  6489.5  100.91  7071.1  100.91
  8251.3  100.95  8659.5  103.01  9189.5  102.71  9269.5  100.91  9528.3  104.51
#Mann= 7 ,-1 , 0
  1935.1     .08       0  4936.5     .04       0    4942     .04       0
  5063.4     .04       0  5068.9     .08       0  7071.1     .05       0
  8251.3     .08       0
#XS Ineff= 3 ,-1
    2500  4936.2    97.8  5057.9    625099.89999    6250    9515     104
Permanent Ineff=
       F       F       F
Bank Sta=4942,5063.4
XS Rating Curve= 0 ,0
Exp/Cntr=0.5,0.3

Type RM Length L Ch R = 1 ,97445.  ,528.4,391,232.8
BEGIN DESCRIPTION:
Equador Drive - D\S - XS 1
END DESCRIPTION:
XS GIS Cut Line= 4
      3061495.79     13887634.08      3061155.47     13885627.93
      3061126.75     13885551.52      3059207.52     13881492.36
#Sta/Elev= 30
  2920.9  104.73  3440.9   103.3  3850.9      99  4120.9   99.91  4910.9   97.89
  4940.9   95.79 4992.69   79.87 5000.69   79.21 5008.78   79.97 5015.67   84.12
  5057.3    95.7  5087.3   98.43  5487.3  100.06  5647.3   97.05  5677.3   98.49
  6167.3   99.19  6247.3   101.5  6487.3   99.63  6967.3  100.87  7027.3   97.79
  7067.3   90.23  7377.3   89.41  7397.3   90.35  7437.3   99.12  7457.3  100.93
  8177.3  102.61  8537.3  101.19  9137.3  102.58  9257.3   100.7  9527.4  104.28
#Mann= 5 ,-1 , 0
  2920.9     .08       0  4910.9     .04       0  5087.3     .08       0
  7067.3     .05       0  8177.3     .08       0
#XS Ineff= 2 , 0
       0                    6255       0     104
Permanent Ineff=
       F       F
#Block Obstruct= 1 ,-1
 6969.16 7490.75   100.9
Bank Sta=4910.9,5087.3
XS Rating Curve= 0 ,0
Exp/Cntr=0.3,0.1

Type RM Length L Ch R = 1 ,97054.0 ,247.4,366,562.2
BEGIN DESCRIPTION:
Cross Section E100-00-00-X70
END DESCRIPTION:
XS GIS Cut Line= 5
       3061638.4     13888271.02      3061513.66     13887797.02
      3061519.82     13885395.06      3061166.63     13885103.85
      3059303.58     13880750.58
#Sta/Elev= 30
  1935.5     107  2295.5     104  4135.6    97.9  4405.6   101.5  4615.6    98.1
  4827.6   100.3  4940.5   98.33  4982.1   82.17  4985.5   77.37    5008   75.66
  5012.3   75.81  5020.8   83.53  5061.2   97.65  6235.4   102.1  6693.6   99.18
  6725.4    96.8  6775.4    87.4  6825.4    98.6  6843.2  100.01    6949   100.5
  7005.4    98.6  7085.4    89.9  7125.4    88.3  7234.4   97.48  7275.4   100.6
  8985.4   102.7  9159.7  100.86  9205.4   102.5  9411.1  101.31 10020.5   104.1
#Mann= 10 ,-1 , 0
  1935.5     .08       0  4940.5     .04       0  5061.2     .08       0
  6693.6     .04       0  6843.2     .08       0    6949     .04       0
  7234.4     .05       0  9159.7     .08       0  9411.1      .1       0
 10020.5     .99       0
#XS Ineff= 2 , 0
       0    3490     104    5589       0     104
Permanent Ineff=
       F       F
#Block Obstruct= 2 ,-1
  6626.2  7275.4   100.6    7276  7276.5      70
Bank Sta=4940.5,5061.2
XS Rating Curve= 0 ,0
Exp/Cntr=0.3,0.1

Type RM Length L Ch R = 1 ,96688.  ,130.1,102,97.3
BEGIN DESCRIPTION:
Hwy 8 South Feeder - U\S - XS 4
-Modified left bank location
END DESCRIPTION:
XS GIS Cut Line= 4
      3061542.33     13887527.71      3061591.85     13886289.63
      3061676.13     13885420.66      3061777.68     13883049.36
#Sta/Elev= 30
  2567.7  104.68  3806.8    98.7  4366.8  100.99  4416.8  100.21  4839.8   100.9
  4889.8   99.46  4909.8   97.28  4939.8   88.94 4973.02    82.8 4978.27   80.45
 4981.26   78.14 4999.01   74.63 5005.34    74.8 5021.73    78.7 5039.14   88.43
 5045.66    97.1 5071.37  100.72  5077.3  100.64 5132.47     101 5224.92     100
 5277.53  101.07 5693.63  100.77 5895.01     100 6101.69   98.94  6399.8  100.06
  6679.8   99.44  6709.8   98.48  6769.8   99.14  6849.8   98.32  7053.3   99.17
#Mann= 4 ,-1 , 0
  2567.7     .08       0  4889.8     .04       0 5045.66     .04       0
 5895.01     .08       0
#XS Ineff= 2 , 0
       0  4779.4     104  5170.1       0     104
Permanent Ineff=
       F       F
Bank Sta=4889.8,5077.3
XS Rating Curve= 0 ,0
Exp/Cntr=0.5,0.3

Type RM Length L Ch R = 1 ,96586.0 ,73,72,67.7
BEGIN DESCRIPTION:
Upstream Section of Bridge/Culvert/Weir
END DESCRIPTION:
XS GIS Cut Line= 6
      3061669.24     13888135.23      3061595.79     13887454.89
      3061631.86     13886365.75      3061697.42     13885859.99
      3061772.35     13885429.15       3061873.9     13883057.85
#Sta/Elev= 30
  1957.9  106.03  2642.2  104.53  3801.9   98.63  4291.9  100.83  4401.9   99.73
  4431.9  100.53  4551.9   99.83  4737.8  101.81  4742.1  100.89  4877.4   101.6
  4896.4    97.7  4917.9   97.48  4926.4   94.33  4937.1   88.66  4958.8   84.74
  4967.8   84.58  4973.6    81.6  4976.9   78.66  4996.5   74.34  5003.3   74.43
  5020.9   77.07  5039.6   88.45  5046.6   98.98  5074.2  101.57  5189.8   100.5
  5229.4   101.8  5870.8   98.94  6929.2   99.43  6989.2  102.13  7052.7  109.13
#Mann= 6 , 1 , 0
  1957.9     .99       0  1957.9     .08       0  4877.4     .04       0
  5074.2     .04       0  5870.8     .08       0  7052.7     .99       0
#XS Ineff= 2 , 0
       0  4879.4     104  5070.1       0     104
Permanent Ineff=
       F       F
Bank Sta=4877.4,5074.2
XS Rating Curve= 0 ,0
Exp/Cntr=0.5,0.3

Type RM Length L Ch R = 3 ,96552.5 ,,,
BEGIN DESCRIPTION:
SAM HOUSTON TOLLWAY-SOUTHBOUND FEEDER
Structure ID: E100-00-00-48
END DESCRIPTION:
Bridge Culvert--1,0,-1,-1, 0
Deck Dist Width WeirC Skew NumUp NumDn MinLoCord MaxHiCord MaxSubmerge Is_Ogee
10,47,2.6,0, 40, 40, , , 0.95, 0, ,,,
  1957.9  2642.2  3612.2  3731.9  3801.9  4011.9  4241.9  4291.9  4401.9  4431.9
  4531.9  4551.9  4679.2  4737.8  4742.1 4802.39  4802.5  4837.5  4877.4 4887.51
  4958.8  5039.6  5060.1  5074.2  5094.5  5120.2  5147.1 5147.21  5189.8  5229.4
  5290.1  5939.2  6559.2  6659.2  6689.2  6929.2  6989.2  7019.2  7029.2  7052.7
     106   104.5   100.1   100.1   100.1   100.1  100.61  100.81  100.53  100.61
  100.87  100.93  101.26  101.79  101.45  101.83  104.63  104.99  105.35  105.44
  105.93  106.14  106.13  106.12   106.1  105.98  105.84  103.04  102.76  102.38
  101.77  100.71    99.7    99.7    98.7    99.4   102.1   104.9   106.8   109.1
     106   104.5   99.78    99.2    98.6     100   100.6   100.8    99.7   100.5
   100.1    99.8   100.7  101.78  100.86  101.57  101.57  101.78  101.57   99.13
   99.63   99.84   99.78  101.54  101.62  101.73  101.24  101.24  100.47  101.77
   101.5    98.6    99.7    99.7    98.7    99.4   102.1   104.9   106.8   109.1
  1957.9  2642.2  3612.2  3731.9  3801.9  4011.9  4241.9  4291.9  4401.9  4431.9
  4531.9  4551.9  4679.2  4737.8  4742.1 4802.39  4802.5  4837.5  4877.4 4887.51
  4958.8  5039.6  5060.1  5074.2  5094.5  5120.2  5147.1 5147.21  5189.8  5229.4
  5290.1  5939.2  6559.2  6659.2  6689.2  6929.2  6989.2  7019.2  7029.2  7052.7
     106   104.5   100.1   100.1   100.1   100.1  100.61  100.81  100.53  100.61
  100.87  100.93  101.26  101.79  101.45  101.83  104.63  104.99  105.35  105.44
  105.93  106.14  106.13  106.12   106.1  105.98  105.84  103.04  102.76  102.38
  101.77  100.71    99.7    99.7    98.7    99.4   102.1   104.9   106.8   109.1
     106   104.5   99.78    99.2    98.6     100   100.6   100.8    99.7   100.5
   100.1    99.8   100.7  101.78  100.86  101.57  101.57  101.78  101.57   99.13
   99.63   99.84   99.78  101.54  101.62  101.73  101.24  101.24  100.47  101.77
   101.5    98.6    99.7    99.7    98.7    99.4   102.1   104.9   106.8   109.1
Pier Skew, UpSta & Num, DnSta & Num=  ,4946.4, 2 ,4946.4, 2 , 0 , 0 , 0 ,,
     1.5     1.5
   85.51  100.57
     1.5     1.5
   85.64   100.7
Pier Skew, UpSta & Num, DnSta & Num=  ,5003.3, 2 ,5003.3, 2 , 0 , 0 , 0 ,,
     1.5     1.5
   73.39  100.78
     1.5     1.5
   73.52  100.91
Abutment Skew #Up #Dn= , 2 , 2
  4887.4    4977
   99.14    78.6
  4887.4    4977
   99.27   78.73
Abutment Skew #Up #Dn= , 2 , 2
  5022.9 5060.19
   78.74   99.83
  5022.9 5060.19
   78.87   99.96
BR Coef= 1 , 1 , 0 ,1.25, 0 ,,,0.8,-1,2,0,
WSPro=,,,, 1 ,,,, 0 ,,,, 0 ,,,,-1 ,-1 ,-1 , 0 , 0 , 0 , 0 , 0
BR U #Sta/Elev= 77
  1957.9     106  2642.2   104.5  2682.3   104.3  3612.2   99.78  3731.9    99.2
  3801.9    98.6  4011.9     100  4236.4  100.59  4241.9   100.6  4291.9   100.8
  4401.9    99.7  4431.9   100.5  4531.9   100.1  4551.9    99.8  4679.2   100.7
  4733.2   101.7  4737.8  101.78  4742.1  100.86  4795.1  101.53  4798.5  101.55
 4802.39  101.57  4802.5  101.57 4802.61  101.57  4837.5  101.78  4852.6   101.7
  4877.4  101.57 4887.51   99.13  4887.6   99.11  4891.1   98.27  4896.4   97.67
  4902.3   97.61  4917.9   97.45  4926.4    94.3  4937.1   88.63  4946.4   86.63
  4951.4   85.86  4958.8   84.71  4967.8   84.55  4973.6   81.57  4976.9   78.63
    4977    78.6  4980.4   77.44  4996.5   74.31  5000.1   74.36  5003.3    74.4
  5020.9   77.04  5022.8   78.68  5022.9   78.74  5039.6   88.42  5042.6   92.93
  5046.6   98.95    5054   99.02 5059.99   99.77  5060.1   99.78  5074.2  101.54
  5094.5  101.62  5120.2  101.73    5122   101.7 5146.99  101.25  5147.1  101.24
 5147.21  101.24  5179.1  100.66  5189.8  100.47  5229.4  101.77  5236.4  101.74
  5290.1   101.5  5870.8   98.91  5939.2    98.6  6559.2    99.7  6619.6    99.7
  6659.2    99.7  6689.2    98.7  6929.2    99.4  6989.2   102.1  7019.2   104.9
  7029.2   106.8  7052.7   109.1
BR U #Mann= 6
  1957.9     .99  1957.9     .08  4877.4    .035  5074.2     .04  5870.8     .08
  7052.7     .99
BR U Banks=4877.4,5074.2
BR D #Sta/Elev= 77
  1957.9     106  2642.2   104.5  2682.3   104.3  3612.2   99.78  3731.9    99.2
  3801.9    98.6  4011.9     100  4236.4  100.59  4241.9   100.6  4291.9   100.8
  4401.9    99.7  4431.9   100.5  4531.9   100.1  4551.9    99.8  4679.2   100.7
  4733.2   101.7  4737.8  101.78  4742.1  100.86  4795.1  101.53  4798.5  101.55
 4802.39  101.57  4802.5  101.57 4802.61  101.57  4837.5  101.78  4852.6   101.7
  4877.4   101.7 4887.51   99.26  4887.6   99.24  4891.1    98.4  4896.4    97.8
  4902.3   97.74  4917.9   97.58  4926.4   94.43  4937.1   88.76  4946.4   86.76
  4951.4   85.99  4958.8   84.84  4967.8   84.68  4973.6    81.7  4976.9   78.76
    4977   78.73  4980.4   77.57  4996.5   74.44  5000.1   74.49  5003.3   74.53
  5020.9   77.17  5022.8   78.81  5022.9   78.87  5039.6   88.55  5042.6   93.06
  5046.6   99.08    5054   99.15 5059.99    99.9  5060.1   99.91  5074.2  101.67
  5094.5  101.62  5120.2  101.73    5122   101.7 5146.99  101.25  5147.1  101.24
 5147.21  101.24  5179.1  100.66  5189.8  100.47  5229.4  101.77  5236.4  101.74
  5290.1   101.5  5870.8   98.91  5939.2    98.6  6559.2    99.7  6619.6    99.7
  6659.2    99.7  6689.2    98.7  6929.2    99.4  6989.2   102.1  7019.2   104.9
  7029.2   106.8  7052.7   109.1
BR D #Mann= 4
  1957.9     .08  4877.4    .035  5074.2     .04  5870.8     .08
BR D Banks=4877.4,5074.2
BC Design=,, 0 ,, 0 ,,,,,,
BC HTab HWMax=109.13
BC Use User HTab Curves=0
BC User HTab FreeFlow(D)= 0

Type RM Length L Ch R = 1 ,96514.0 ,55.2,55,52
BEGIN DESCRIPTION:
Downstream Section of Bridge/Culvert/Weir
END DESCRIPTION:
XS GIS Cut Line= 6
      3061736.16     13888143.91      3061662.93     13887465.67
      3061698.88     13886380.09      3061764.18     13885876.39
      3061839.32     13885444.28      3061940.96     13883071.04
#Sta/Elev= 30
  1957.9  106.03  2642.2  104.53  3801.9   98.63  4291.9  100.83  4401.9   99.73
  4431.9  100.53  4551.9   99.83  4737.8  101.81  4742.1  100.89  4877.4  101.83
  4896.4   97.93  4917.9   97.71  4926.4   94.56  4937.1   88.89  4958.8   84.97
  4967.8   84.81  4973.6   81.83  4976.9   78.89  4996.5   74.57  5003.3   74.66
  5020.9    77.3  5039.6   88.68  5046.6   99.21  5074.2   101.8  5189.8   100.5
  5229.4   101.8  5870.8   98.94  6929.2   99.43  6989.2  102.13  7052.7  109.13
#Mann= 5 ,-1 , 0
  1957.9     .08       0  4877.4     .04       0  5074.2     .04       0
  5870.8     .08       0  7052.7     .99       0
#XS Ineff= 2 , 0
       0  4879.4     104  5070.1       0     104
Permanent Ineff=
       F       F
Bank Sta=4877.4,5074.2
XS Rating Curve= 0 ,0
Exp/Cntr=0.5,0.3

Type RM Length L Ch R = 1 ,96459.0 ,160,161,161.1
BEGIN DESCRIPTION:
Upstream Section of Bridge/Culvert/Weir
END DESCRIPTION:
XS GIS Cut Line= 4
      3061702.68     13887070.73      3061716.38     13886484.67
       3061900.2     13885353.05      3061958.42     13883186.21
#Sta/Elev= 30
  3052.9  109.85  3063.3  109.75  3393.3  113.75  3523.3  111.05  3659.5  104.05
  3889.5  105.65  3949.5  100.75  4069.5  100.65  4089.5  101.35  4139.5  109.75
  4649.5  107.95  4710.8  118.01  4808.9  111.41  4903.3  108.69  4925.8   97.25
  4968.7   87.59    4973   81.84  4977.3   79.45  4993.5   75.54  5018.4   77.65
    5022   82.49  5091.2     100  5101.1  104.58  5264.6  106.27  5613.3  104.29
    6486  100.95    6676  106.15    6736   98.55    6916   99.35  6963.6  113.65
#Mann= 6 , 1 , 0
  3052.9     .99       0  3063.3     .08       0  4903.3     .04       0
  5101.1     .12       0  5613.3     .08       0  6963.6     .99       0
#XS Ineff= 2 , 0
       0  4909.3     109  5099.9       0   104.5
Permanent Ineff=
       F       F
Bank Sta=4903.3,5101.1
XS Rating Curve= 0 ,0
Exp/Cntr=0.5,0.3

Type RM Length L Ch R = 3 ,96380.5 ,,,
BEGIN DESCRIPTION:
SAM HOUSTON TOLLWAY MAIN LANES
Structure ID: E100-00-00-47a
END DESCRIPTION:
Bridge Culvert--1,0,-1,-1, 0
Deck Dist Width WeirC Skew NumUp NumDn MinLoCord MaxHiCord MaxSubmerge Is_Ogee
10,137,2.6,0, 60, 60, 106.4, , 0.95, 0, ,,,
  3052.9  3153.3  3273.3  3283.3  3393.3  3453.3  3463.3  3523.3  3583.3  3659.5
  3689.5  3849.5  3878.7  3888.7  3898.7  3919.5  3938.7  3949.5  3958.7  4059.5
  4078.7  4089.5  4108.7  4119.5  4129.5  4148.7  4158.7  4619.5  4649.5 4710.49
  4710.6  4710.8  4808.9  4865.9  4903.3  4911.3  4913.3  5009.5  5091.2  5101.1
  5194.2    5264 5264.11  5264.6  5728.9    5956    6366    6486    6576  6669.4
  6679.4    6696    6706    6716    6736  6749.3    6776    6916    6936  6963.6
     110  112.04  114.49  114.69  116.93  118.15  118.36  119.58  120.53  121.24
  121.53  123.03   123.3   122.1   119.9  112.36   105.4  102.56     101  101.42
   101.5  103.27   107.6  111.38  114.88   120.9   122.5  118.88  118.64  118.16
  120.96  120.96  118.66  117.31  116.46  116.28  116.24  113.93  112.25  112.06
  110.44  109.23  106.43  106.42   108.4  112.67  120.39  122.65  124.34   126.1
     124  119.39  116.36  113.32  107.24   103.2    99.4    99.5   104.9   113.8
  109.99  111.89  113.39  113.09  113.89  112.29  112.49  111.19  107.49  104.19
  105.29  104.99  105.57  105.77  105.42  104.59  102.48  100.89  100.84  101.29
  100.88  101.49  105.59  107.89  109.29  109.84  109.79  107.49  108.09   118.1
  118.12  118.15  111.55  110.25  108.83  105.15  104.83  102.52  100.84  104.72
  104.18  106.39  106.39  106.41  103.78  102.49  102.39  101.09  102.19  105.89
  106.19  105.09  103.59  101.19   98.69   98.92   99.39   99.49  104.89  113.79
  3052.9  3153.3  3273.3  3283.3  3353.3  3393.3  3453.3  3463.3  3523.3  3583.3
  3659.5  3689.5  3849.5  3878.7  3888.7  3898.7  3919.5  3938.7  3949.5  3958.7
  4059.5  4078.7  4089.5  4108.7  4119.5  4129.5  4148.7  4158.7  4619.5  4649.5
 4710.49  4710.6  4710.8  4808.9  4865.9  4903.3  4911.3  4913.3  5009.5  5091.2
  5101.1  5194.2    5264 5264.11  5728.9    5956    6366    6486    6576  6669.4
  6679.4    6696    6706    6716    6736  6749.3    6776    6916    6936  6963.6
  110.25  112.15  114.49  114.69  116.12  116.93  118.15  118.36  119.58  120.53
  121.24  121.53  123.03   123.3   122.1   119.9  112.36   105.4  102.56   101.1
  101.55   101.5  103.27   107.6  111.38  114.88   120.9   122.5  118.88  118.64
  118.36  120.96  120.96  118.66  117.31  116.46  116.28  116.24  113.93  112.25
  112.06  110.44  109.23  106.65   108.4  112.67  120.39  122.65  124.34   126.1
     124  119.39  116.36  113.32  107.24   103.2   99.65   99.75  105.15  114.05
  110.25  112.15  113.65  113.35  114.25  114.15  112.55  112.75  111.45  107.75
  104.45  105.55  105.25  105.83  106.03  105.68  104.85  102.74  101.15   101.1
  101.55  101.14  101.75  105.85  108.15  109.55   110.1  110.05  107.75  108.35
  118.36  118.38  118.41  111.81  110.51  109.09  105.41  105.09  102.78   101.1
  104.98  104.44  106.65  106.65  104.04  102.75  102.65  101.35  102.45  106.15
  106.45  105.35  103.85  101.45   98.95   99.18   99.65   99.75  105.15  114.05
Pier Skew, UpSta & Num, DnSta & Num=  ,4973, 2 ,4973, 2 , 0 , 0 , 0 ,,
     1.5     1.5
   80.56  104.42
     1.5     1.5
   80.82  104.68
Pier Skew, UpSta & Num, DnSta & Num=  ,5032.7, 2 ,5032.7, 2 , 0 , 0 , 0 ,,
     1.5     1.5
   83.75  103.06
     1.5     1.5
   84.01  103.32
Abutment Skew #Up #Dn= , 2 , 2
  4911.1    4981
  105.15   78.26
  4911.1    4981
  105.41   78.52
Abutment Skew #Up #Dn= , 2 , 2
    5019 5098.99
   78.47  103.65
    5019 5098.99
   78.73  103.91
BR Coef= 1 , 1 , 0 ,1.25, 0 ,,,0.8,0,2,0,
WSPro=,,,, 1 ,,,, 0 ,,,, 0 ,,,,-1 ,-1 ,-1 , 0 , 0 , 0 , 0 , 0
BR U #Sta/Elev= 127
  3052.9  109.99  3063.3  109.89  3153.3  111.89  3213.3  112.69  3253.3  112.89
  3273.3  113.39  3283.3  113.09  3353.3  113.99  3383.3  113.69  3393.3  113.89
  3403.3  113.49  3433.3  113.09  3453.3  112.29  3463.3  112.49  3513.3  111.19
  3523.3  111.19  3558.7  109.21  3573.3  108.39  3583.3  107.49  3603.3  106.79
  3649.5  104.39  3659.5  104.19  3689.5  105.29  3719.5  105.29  3739.5  105.49
  3749.5  104.99  3829.5  105.29  3849.5  104.99  3878.7  105.57  3888.7  105.77
  3889.5  105.79  3898.7  105.42  3919.5  104.59  3938.7  102.48  3939.5  102.39
  3948.7  101.01  3949.5  100.89  3958.7  100.84  3969.5  100.79  4059.5  101.29
  4069.5  100.79  4078.7  100.88  4079.5  100.89  4088.7  101.44  4089.5  101.49
  4098.7  103.45  4108.7  105.59  4119.5  107.89  4129.5  109.29  4138.7  109.84
  4139.5  109.89  4148.7  109.84  4158.7  109.79  4619.5  107.49  4649.5  108.09
 4710.49   118.1  4710.6  118.12 4710.71  118.14  4710.8  118.15  4710.9  118.14
  4763.1  114.63  4808.9  111.55  4815.5   111.4  4865.8  110.25  4865.9  110.25
  4903.3  108.83 4911.21  105.19  4911.3  105.15  4913.3  104.23  4919.3  100.95
  4925.8   97.39  4948.9   92.45  4968.7   87.73    4972   83.53  4972.9   82.39
    4973   81.98  4977.3   79.59  4979.9   79.22  4980.9   78.32    4981   78.26
    4983   77.02  4993.5   75.68  5009.5   77.04  5018.4   77.79  5018.9   78.33
    5019   78.47    5022   82.63  5032.7   84.91  5047.5   88.48  5076.4   96.83
  5091.2  100.14 5098.79  103.65  5098.9   103.7    5099  103.75  5101.1  104.72
  5142.3  104.64  5143.9  104.63  5194.2  104.18  5200.2  104.37 5263.89  106.39
    5264  106.39 5264.11  106.39  5264.5  106.41  5264.6  106.41  5613.3  104.43
  5728.9  103.78    5956  102.49    6366  102.39    6486  101.09    6576  102.19
    6666  105.69  6669.4  105.89    6676  106.29  6679.4  106.19    6686  105.99
  6689.4  105.68    6696  105.09    6706  103.59    6716  101.19    6726   99.69
    6736   98.69  6749.3   98.92    6776   99.39    6916   99.49    6926  101.89
    6936  104.89  6963.6  113.79
BR U #Mann= 6
  3052.9     .99  3063.3     .08  4903.3    .035  5101.1     .12  5613.3     .08
  6963.6     .99
BR U Banks=4903.3,5101.1
BR D #Sta/Elev= 127
  3052.9  110.25  3063.3  110.15  3153.3  112.15  3213.3  112.95  3253.3  113.15
  3273.3  113.65  3283.3  113.35  3353.3  114.25  3383.3  113.95  3393.3  114.15
  3403.3  113.75  3433.3  113.35  3453.3  112.55  3463.3  112.75  3513.3  111.45
  3523.3  111.45  3558.7  109.47  3573.3  108.65  3583.3  107.75  3603.3  107.05
  3649.5  104.65  3659.5  104.45  3689.5  105.55  3719.5  105.55  3739.5  105.75
  3749.5  105.25  3829.5  105.55  3849.5  105.25  3878.7  105.83  3888.7  106.03
  3889.5  106.05  3898.7  105.68  3919.5  104.85  3938.7  102.74  3939.5  102.65
  3948.7  101.27  3949.5  101.15  3958.7   101.1  3969.5  101.05  4059.5  101.55
  4069.5  101.05  4078.7  101.14  4079.5  101.15  4088.7   101.7  4089.5  101.75
  4098.7  103.71  4108.7  105.85  4119.5  108.15  4129.5  109.55  4138.7   110.1
  4139.5  110.15  4148.7   110.1  4158.7  110.05  4619.5  107.75  4649.5  108.35
 4710.49  118.36  4710.6  118.38 4710.71   118.4  4710.8  118.41  4710.9   118.4
  4763.1  114.89  4808.9  111.81  4815.5  111.66  4865.8  110.51  4865.9  110.51
  4903.3  109.09 4911.21  105.45  4911.3  105.41  4913.3  104.49  4919.3  101.21
  4925.8   97.65  4948.9   92.71  4968.7   87.99    4972   83.79  4972.9   82.65
    4973   82.24  4977.3   79.85  4979.9   79.48  4980.9   78.58    4981   78.52
    4983   77.28  4993.5   75.94  5009.5    77.3  5018.4   78.05  5018.9   78.59
    5019   78.73    5022   82.89  5032.7   85.17  5047.5   88.74  5076.4   97.09
  5091.2   100.4 5098.79  103.91  5098.9  103.96    5099  104.01  5101.1  104.98
  5142.3   104.9  5143.9  104.89  5194.2  104.44  5200.2  104.63 5263.89  106.65
    5264  106.65 5264.11  106.65  5264.5  106.67  5264.6  106.67  5613.3  104.69
  5728.9  104.04    5956  102.75    6366  102.65    6486  101.35    6576  102.45
    6666  105.95  6669.4  106.15    6676  106.55  6679.4  106.45    6686  106.25
  6689.4  105.94    6696  105.35    6706  103.85    6716  101.45    6726   99.95
    6736   98.95  6749.3   99.18    6776   99.65    6916   99.75    6926  102.15
    6936  105.15  6963.6  114.05
BR D #Mann= 6
  3052.9     .99  3063.3     .08  4903.3    .035  5101.1     .12  5613.3     .08
  6963.6     .99
BR D Banks=4903.3,5101.1
BC Design=,, 0 ,, 0 ,,,,,,
BC HTab HWMax=118.01
BC Use User HTab Curves=0
BC User HTab FreeFlow(D)= 0

Type RM Length L Ch R = 1 ,96298.0 ,52,54,55.9
BEGIN DESCRIPTION:
Downstream Section of Bridge/Culvert/Weir
END DESCRIPTION:
XS GIS Cut Line= 4
      3061832.57     13887066.82      3061877.19     13886491.15
      3062060.98     13885359.68      3062119.37      13883186.8
#Sta/Elev= 30
  3052.9  110.29  3063.3  110.19  3393.3  114.19  3523.3  111.49  3659.5  104.49
  3889.5  106.09  3949.5  101.19  4069.5  101.09  4089.5  101.79  4139.5  110.19
  4649.5  108.39  4710.8  118.45  4808.9  111.85  4903.3  109.13  4925.8   97.69
  4968.7   88.03    4973   82.28  4977.3   79.89  4993.5   75.98  5018.4   78.09
    5022   82.93  5091.2  100.44  5101.1  105.02  5264.6  106.71  5613.3  104.73
    6486  101.39    6676  106.59    6736   98.99    6916   99.79  6963.6  114.09
#Mann= 6 , 1 , 0
  3052.9     .99       0  3063.3     .08       0  4903.3     .04       0
  5101.1     .12       0  5613.3     .08       0  6963.6     .99       0
#XS Ineff= 2 , 0
       0  4909.3     109  5099.9       0   104.5
Permanent Ineff=
       F       F
Bank Sta=4903.3,5101.1
XS Rating Curve= 0 ,0
Exp/Cntr=0.5,0.3

Type RM Length L Ch R = 1 ,96244.0 ,67.6,68,69
BEGIN DESCRIPTION:
Upstream Section of Bridge/Culvert/Weir
END DESCRIPTION:
XS GIS Cut Line= 4
      3061773.25     13888068.17      3061876.51     13886665.54
      3062112.03     13885332.86      3062192.45     13883557.87
#Sta/Elev= 30
  2052.3  106.06  2846.8  106.69  3062.3  106.86  3458.7  110.26  3668.7  108.26
  3888.7  107.86  3908.7  106.26  3938.7  101.06  4015.7  101.36  4078.7  100.86
  4118.7  107.26  4138.7  107.76  4711.7  101.35    4895   103.3  4919.9   96.75
  4955.1   89.42    4969   84.97    4980   83.54  4991.3   76.72  5004.3    76.2
  5010.9   77.57    5018   83.69  5092.7  103.32  5276.7  102.39  5278.3  101.63
  5512.1  102.46    5616  104.02  5912.1  108.56  6372.1  107.66  6588.9  103.16
#Mann= 7 ,-1 , 0
  2052.3     .08       0  2846.8     .05       0  4015.7     .12       0
    4895     .04       0  5092.7     .12       0    5616     .08       0
  6588.9     .99       0
#XS Ineff= 2 , 0
       0  4898.4     102  5088.9       0   101.9
Permanent Ineff=
       F       F
Bank Sta=4895,5092.7
XS Rating Curve= 0 ,0
Exp/Cntr=0.5,0.3
